--- GldCrk.prj (project) ---

Proj Title=GldCrk
Current Plan=p02
Default Exp/Contr=0,0
English Units
Geom File=g01
Geom File=c:\temp\GldCrk.g02
Flow File=f01
Plan File=p01
Plan File=p02
BEGIN DESCRIPTION:
END DESCRIPTION:
DSS Export Rating Curves= 0
DSS Export Rating Curve Sorted= 0
DSS Export Volume Flow Curves= 0
DXF OffsetX= 0
DXF OffsetY= 0
DXF ScaleX= 0
DXF ScaleY= 0

--- GldCrk.p01 (plan) ---

Plan Title=Floodplain
Program Version=4.00
Geom File=g01
Flow File=f01
K Sum by GR=0
Std Step Tol=0.01
Critical Tol=0.01
Num of Std Step Trials=20
Max Error Tol=0.3
Flow Tol Ratio=0.001
Split Flow NTrial=30
Split Flow Tol=0.02
Split Flow Ratio=0.02
Log Output Level=0
Friction Slope Method=1
Unsteady Friction Slope Method=2
Unsteady Bridges Friction Slope Method=1
Global Log Level=0
CheckData=False
Run HTab=0
Run UNet=0
Run PostProcess=0
UNET Theta=0
UNET Theta Warmup=0
UNET ZTol=0
UNET ZSATol=0
UNET MxIter=0
UNET MaxInSteps=0
UNET DtIC=0
UNET DtMin=0
UNET MaxCRTS=0
UNET WFStab=0
UNET SFStab=0
UNET WFX=0
UNET SFX=0
UNET DSS MLevel=0
UNET DZMax Abort=0
UNET Convert EG Bridges=0
UNET Use Existing IB Tables=0
UNET Froude Limit=0
UNET Froude Power=0
Write IC File=0
Echo Input=False
Echo Output=False
Write Detailed=0

--- GldCrk.f01 (steady flow) ---

Flow Title=NFF Regression Equation
Program Version=4.00
Number of Profiles=1
Profile Names=P100yr
River Rch & RM=GldCrk,Main      ,92150.4
2469.586
River Rch & RM=GldCrk,Main      ,91148.9
2633.356
River Rch & RM=GldCrk,Main      ,83606.9
2806.819
River Rch & RM=GldCrk,Main      ,73696.5
3101.186
River Rch & RM=GldCrk,Main      ,73179.3
3849.136
River Rch & RM=GldCrk,Main      ,66812.1
3960.190
River Rch & RM=GldCrk,Main      ,56488
4377.581
River Rch & RM=GldCrk,Main      ,43716.9
4837.345
River Rch & RM=GldCrk,Main      ,31729.8
5141.320
River Rch & RM=GldCrk,Main      ,31393.5
6895.091
River Rch & RM=GldCrk,Main      ,23321.4
7420.569
Boundary for River Rch & Prof#=GldCrk,Main      ,1
Up Type=0
Dn Type=3
Dn Slope=0.023025

--- GldCrk.g01 (geometry) ---

Geom Title=USGS 3m DEM
Program Version=4.10

River Reach=GldCrk          ,Main
Reach XY= 30
     1944469.304      238610.482     1945753.305      242802.974
     1947115.706      244109.514     1948923.731      243892.497
        1949779.      244596.401     1953548.648      249835.659
     1953479.617      252754.671     1951734.891      254248.655
     1953360.076      256283.443     1952736.215      257912.999
     1951031.951      257784.745     1951134.815      258995.683
     1952736.378      260560.787     1951661.278      264290.175
     1950435.054      265016.461     1950694.724      267389.386
     1952305.891      268324.782     1952244.191      269546.464
     1954321.819      270503.033     1952447.448      276682.473
     1953216.847      277715.735      1955856.17      278184.485
     1958020.232      281968.339     1959419.972      282921.464
     1959847.055      285000.891     1959186.899      286542.558
     1960952.591      292068.579     1964452.524      293573.808
     1966748.097      297377.193     1964816.226      302331.281

Type RM Length L Ch R = 1 ,92150.4 ,652.6,689.8,727
XS GIS Cut Line= 3
     1944533.978      239021.103     1944704.634      238324.388
     1945337.157      238202.268
#Sta/Elev= 30
       0 2851.59    59.8  2861.9   129.5  2861.5   139.5 2860.72   179.3 2851.49
   229.1 2835.95   249.1 2832.09   404.2 2824.73   418.4 2824.69   419.2 2824.71
   428.4  2824.9   468.2 2830.98   508.1 2843.07   587.8 2846.91   647.6 2855.12
   687.4 2865.03   717.3 2865.58     747 2870.32   856.1 2878.77   955.2 2893.65
  1004.7 2899.64  1034.5 2900.83  1064.2 2898.84  1113.7 2891.84  1133.6 2886.95
  1183.1 2882.52    1193 2883.06  1252.5  2897.6  1292.1 2904.01  1361.5 2912.39
#Mann= 3 , 0 , 0
       0      .1       0   404.2    .045       0   419.2      .1       0
Bank Sta=404.2,419.2
XS Rating Curve= 0 ,0
Exp/Cntr=0.3,0.1

Type RM Length L Ch R = 1 ,91460.7 ,312.2,311.7,311.2
XS GIS Cut Line= 4
     1944510.257       239044.87     1944791.021      238949.523
     1945294.511      239104.672     1945441.005      238937.727
#Sta/Elev= 30
       0 2849.54    59.3 2846.23   128.5 2844.86     168 2842.27   197.7 2842.01
   207.6  2840.2   247.1 2837.39   276.8 2834.29   306.4 2829.67   346.2 2825.08
   366.1 2822.01     376 2819.88   425.7 2814.88   455.6 2813.22   525.2 2812.55
   532.4 2812.56   547.4 2813.28   634.5 2813.68   654.4 2814.52   694.1  2818.3
     714 2821.35   773.7 2828.56   793.5 2831.17   803.5 2833.56   823.4 2836.52
     891 2840.21   977.9 2836.18  1006.8 2833.57  1026.2 2834.24  1045.5  2836.7
#Mann= 3 , 0 , 0
       0      .1       0   532.4    .045       0   547.4      .1       0
Bank Sta=532.4,547.4
XS Rating Curve= 0 ,0
Exp/Cntr=0.3,0.1

Type RM Length L Ch R = 1 ,91148.9 ,326.4,332.3,338.1
XS GIS Cut Line= 3
     1944394.071      239149.096     1945296.573       239407.09
     1945371.977      239412.231
#Sta/Elev= 30
       0 2853.88    49.9 2842.52    69.9 2836.06   129.8 2822.84   139.8 2820.43
   149.8 2817.08   199.7 2807.36   209.7 2806.25   229.7 2805.46   319.5 2805.68
   379.5 2806.82   419.4 2808.13   469.3  2808.9   519.3 2808.93   659.5 2807.85
   674.5 2808.73     709  2810.7   738.9 2811.84   778.9 2813.89   818.8 2814.64
   838.8  2815.4   888.7 2815.91   918.7 2815.82   928.7 2816.28   938.6 2816.94
   948.1  2818.3   985.9 2824.56   995.3  2826.7  1004.8 2828.38  1014.2  2829.4
#Mann= 3 , 0 , 0
       0      .1       0   659.5    .045       0   674.5      .1       0
Bank Sta=659.5,674.5
XS Rating Curve= 0 ,0
Exp/Cntr=0.3,0.1

Type RM Length L Ch R = 1 ,90816.8 ,452.8,441.4,430
XS GIS Cut Line= 2
     1944400.906      239251.613     1945281.171      239860.137
#Sta/Elev= 30
       0 2841.58      50 2832.45      60 2829.25      70  2824.9      90 2818.93
     120 2811.99     140 2806.75     150 2805.16     160  2804.3     180 2803.48
     370 2804.21   500.1 2803.82   620.1 2800.92   633.4    2801   648.4 2801.17
   700.1 2804.67   710.1 2805.77   730.1 2809.27   760.1 2816.37   780.1 2821.98
   810.1 2828.38   830.1 2830.88   850.1 2835.42   860.1 2837.96   870.1 2841.53
   950.1 2860.02   970.1  2866.1   990.1 2868.79  1060.1 2886.81  1070.1 2888.57
#Mann= 3 , 0 , 0
       0      .1       0   633.4    .045       0   648.4      .1       0
Bank Sta=633.4,648.4
XS Rating Curve= 0 ,0
Exp/Cntr=0.3,0.1

Type RM Length L Ch R = 1 ,90375.4 ,520.6,502.1,483.6
XS GIS Cut Line= 2
     1944112.719      239909.144     1945244.481      239950.274
#Sta/Elev= 30
       0 2891.68     9.9 2889.31    29.8 2880.46    99.3 2858.07   119.2  2848.3
   178.8    2830   198.7 2821.27   238.4 2811.08   278.2 2802.35   347.7 2797.87
   521.6 2797.57   536.6 2797.47     606 2797.28   625.9 2798.02   655.7 2800.93
   715.3 2807.98   725.2 2809.76     755 2818.56   764.9 2823.33   834.5 2839.77
   844.4 2844.41   884.2 2853.44     914 2861.07   923.9 2865.95   963.6 2876.15
   993.4 2880.07  1003.4 2882.25    1053  2887.5  1092.8    2890  1132.5 2889.86
#Mann= 3 , 0 , 0
       0      .1       0   521.6    .045       0   536.6      .1       0
Bank Sta=521.6,536.6
XS Rating Curve= 0 ,0
Exp/Cntr=0.3,0.1

Type RM Length L Ch R = 1 ,89873.1 ,258.2,241.1,224.1
XS GIS Cut Line= 3
     1944402.045      240749.783     1945017.146      240141.516
     1945279.635      240038.632
#Sta/Elev= 30
       0 2886.35    29.8 2883.53    79.6 2872.86   129.3 2858.42   149.2 2855.64
   159.1 2852.83   218.8 2833.26   268.5 2822.14   298.3 2817.52   318.2 2811.65
   338.1 2803.83   367.9  2795.8   407.7 2791.69   427.6 2791.01   437.5  2791.5
   556.8 2797.07   636.4 2796.94   656.3 2798.55   666.2  2802.1   745.8 2816.64
   795.5 2828.49   825.3 2833.75   874.8 2848.51   884.5 2853.31   894.2 2856.37
   962.3 2874.27     972 2877.63  1040.1  2884.7    1079 2886.49    1147 2887.64
#Mann= 3 , 0 , 0
       0      .1       0   407.7    .045       0   437.5      .1       0
Bank Sta=407.7,437.5
XS Rating Curve= 0 ,0
Exp/Cntr=0.3,0.1

Type RM Length L Ch R = 1 ,89631.8 ,468.2,498.6,528.9
XS GIS Cut Line= 3
      1944987.53      240745.227     1945019.424      240203.026
     1945383.929      240127.847
#Sta/Elev= 30
       0 2843.36     9.9  2843.2    88.9 2815.46    98.8 2814.87   108.6 2812.01
   138.2 2799.89   148.1 2797.91   276.5 2790.59   295.9 2789.96   306.1 2789.63
   310.9 2789.71   325.9 2791.03   365.4 2802.82   385.1  2804.9   414.8 2810.38
   454.3 2816.68     474 2818.27   503.6 2823.57   543.1  2833.2   552.9 2835.95
   562.7 2840.03   592.1 2847.92   641.1  2859.4     690 2861.41   748.8 2867.49
   778.2 2872.84     788 2875.35   807.6 2881.61   827.2 2882.82   915.3 2884.07
#Mann= 3 , 0 , 0
       0      .1       0   295.9    .045       0   310.9      .1       0
Bank Sta=295.9,310.9
XS Rating Curve= 0 ,0
Exp/Cntr=0.3,0.1

Type RM Length L Ch R = 1 ,89133.2 ,305.6,307,308.4
XS GIS Cut Line= 2
     1944833.041      240893.205     1945658.444      240741.734
#Sta/Elev= 30
       0 2868.86      40 2873.22      50 2873.75    89.9 2872.56   109.9 2869.88
   199.8 2839.49   209.8 2834.87   219.8 2828.37   249.8 2817.17   269.7 2810.64
   289.7 2805.34   299.7 2801.94   369.6 2793.43   379.6 2790.23   389.6 2789.16
   399.6 2788.98   411.5 2789.29   426.5 2790.27   599.4 2801.38   609.4 2802.49
   629.4 2807.18   659.4 2812.82   689.3 2819.56   699.3 2822.94   709.3 2827.25
   739.3 2836.94   769.2 2848.02   779.2 2852.45   789.2 2858.94   839.2 2875.88
#Mann= 3 , 0 , 0
       0      .1       0   411.5    .045       0   426.5      .1       0
Bank Sta=411.5,426.5
XS Rating Curve= 0 ,0
Exp/Cntr=0.3,0.1

Type RM Length L Ch R = 1 ,88826.2 ,347.5,345.8,344
XS GIS Cut Line= 2
      1944891.43      241168.132     1945704.439      241069.252
#Sta/Elev= 30
       0 2844.87      20 2848.54      30 2849.01      40 2848.17    69.9 2844.17
   109.9 2838.16   139.8 2833.49   189.8 2822.69   219.7 2815.89   229.7 2813.04
   239.7  2809.2   249.7 2807.22   309.6 2797.56   319.6 2795.22   371.9 2788.79
   379.5 2788.47   386.9  2788.6   469.4 2793.78   479.4 2794.97   549.3 2800.28
   559.3  2801.9   639.2 2809.03   649.2 2810.68   719.1 2817.66   729.1 2819.74
   759.1  2823.7     779 2827.61     799 2832.39     809 2836.78     819  2840.3
#Mann= 3 , 0 , 0
       0      .1       0   371.9    .045       0   386.9      .1       0
Bank Sta=371.9,386.9
XS Rating Curve= 0 ,0
Exp/Cntr=0.3,0.1

Type RM Length L Ch R = 1 ,88480.3 ,401,400,395.9
XS GIS Cut Line= 3
     1944928.159      241541.757     1945329.919      241462.537
     1945730.984      241379.751
#Sta/Elev= 30
       0 2881.22      40 2882.94    49.9 2882.69    69.9 2879.51    99.9 2872.68
   109.9 2870.25   119.8 2865.43   139.8 2859.28   169.8 2847.95   189.8 2841.26
   199.8 2835.53   209.7 2831.12   229.7 2824.35   269.7 2815.87   349.6 2797.64
   369.6 2791.68   389.5 2788.35     402 2787.44   409.5 2787.29     417  2787.3
   439.5 2787.62   529.4 2791.95   539.3 2792.96   579.3 2794.04   609.3 2795.81
   689.2 2807.23   709.2 2811.88   769.1 2822.57     789  2828.1     819 2833.48
#Mann= 3 , 0 , 0
       0      .1       0     402    .045       0     417      .1       0
Bank Sta=402,417
XS Rating Curve= 0 ,0
Exp/Cntr=0.3,0.1

Type RM Length L Ch R = 1 ,88080.3 ,331,331.7,335.7
XS GIS Cut Line= 3
     1945069.141      241913.396      1945517.17      241805.085
     1945888.954      241656.372
#Sta/Elev= 30
       0 2873.79    19.6 2869.82    58.8 2863.38    68.6 2860.56   117.7 2852.02
   137.3 2847.86   156.9 2842.02   225.6 2828.31   235.4 2825.08     304 2813.62
   323.6 2809.18   372.7 2801.47   382.5 2799.46   402.1 2793.27   421.7 2789.62
   431.5 2788.12   451.1  2787.3   453.4  2787.3   468.4 2787.32   558.6 2793.92
   568.4  2795.3   617.2 2799.53     666  2805.5   724.6  2810.5   734.4 2811.87
   763.7 2818.01     793 2823.28   812.5 2825.58   841.8 2827.84   861.4 2831.16
#Mann= 3 , 0 , 0
       0      .1       0   453.4    .045       0   468.4      .1       0
Bank Sta=453.4,468.4
XS Rating Curve= 0 ,0
Exp/Cntr=0.3,0.1

Type RM Length L Ch R = 1 ,87748.6 ,566.8,558.3,549.8
XS GIS Cut Line= 2
     1944797.876      242286.162      1945928.89      242022.964
#Sta/Elev= 30
       0 2845.81    99.2  2859.3   168.7 2863.67   218.4 2864.77   238.2 2861.59
     258 2855.84     268 2851.78   287.8 2848.51   307.7 2845.85   416.8 2836.34
   436.7 2832.06   506.2 2821.97   585.6 2807.14   595.5 2804.14   605.4 2802.54
     665 2794.71   684.8 2791.12   714.6 2787.84   734.5  2787.3   746.8  2787.3
   761.8 2787.33   784.1 2788.12   903.2 2796.68     923 2798.47   972.7 2805.59
  1002.4 2810.67  1022.3 2816.34  1081.8 2829.05  1101.7 2836.41  1161.2 2848.81
#Mann= 3 , 0 , 0
       0      .1       0   746.8    .045       0   761.8      .1       0
Bank Sta=746.8,761.8
XS Rating Curve= 0 ,0
Exp/Cntr=0.3,0.1

Type RM Length L Ch R = 1 ,87189.9 ,312.8,309.6,306.9
XS GIS Cut Line= 2
     1945085.783      242981.937     1945976.847      242358.818
#Sta/Elev= 30
       0 2864.61      10 2864.49    79.8 2856.84   159.6 2852.63   199.5 2848.22
   249.4 2839.53   289.3 2828.91   309.2 2825.32   349.1 2825.36     389 2820.76
   448.9 2816.32   478.8 2811.82   528.7 2806.15   568.6 2799.91   628.4 2791.96
   671.6  2787.4   678.3  2787.3   686.6  2787.3   718.2 2787.32   738.2 2789.25
   758.1 2794.69   788.1  2801.5     818 2806.98   857.9 2815.88   897.8 2821.96
   937.7 2826.86   957.6 2830.78  1037.4 2843.59  1057.4 2848.44  1087.3 2853.38
#Mann= 3 , 0 , 0
       0      .1       0   671.6    .045       0   686.6      .1       0
Bank Sta=671.6,686.6
XS Rating Curve= 0 ,0
Exp/Cntr=0.3,0.1

Type RM Length L Ch R = 1 ,86880.3 ,273.9,275.3,276.1
XS GIS Cut Line= 3
     1945502.941      243134.325     1945801.684      242854.652
     1946108.825      242581.449
#Sta/Elev= 30
       0 2848.26    39.9 2845.03    49.9 2843.63    69.9 2837.79    79.8 2836.24
   109.8  2829.8   159.7 2821.95   169.7 2819.61   259.5 2807.23   269.5 2805.32
   279.5 2802.43   309.4 2796.33   319.4 2793.78   329.4 2790.64   339.4 2788.31
   349.3 2787.34   359.3  2787.3   458.2  2787.3   477.7 2787.78   516.9 2791.91
   585.4 2802.49     605 2806.57   614.8 2808.14   634.3 2809.89     693 2819.63
     742  2828.4   761.6 2833.11   771.4 2834.39   781.1 2836.43   820.3 2849.44
#Mann= 3 , 0 , 0
       0      .1       0   359.3    .045       0   458.2      .1       0
Bank Sta=359.3,458.2
XS Rating Curve= 0 ,0
Exp/Cntr=0.3,0.1

Type RM Length L Ch R = 1 ,86605   ,788.4,782.2,776
XS GIS Cut Line= 2
     1945292.043      243634.304     1946336.975      242758.061
#Sta/Elev= 30
       0 2819.88    69.7 2817.39    89.6 2815.42   119.4 2809.38   129.4 2809.36
   169.2  2805.6   199.1  2807.5   258.8 2814.54   278.7  2814.1   318.5 2816.84
   338.4 2815.33   418.1  2817.9     438 2816.93   467.8 2817.61   507.7 2816.82
   557.4 2818.41     647 2814.36   726.6 2804.77   826.2 2788.34     856  2787.3
  1025.3  2787.3  1055.1  2788.8  1154.7 2812.24  1164.6 2815.47  1184.5 2825.52
  1274.1 2865.84  1284.1 2871.17    1304 2874.66  1333.8 2882.29  1363.7 2886.22
#Mann= 3 , 0 , 0
       0      .1       0     856    .045       0  1025.3      .1       0
Bank Sta=856,1025.3
XS Rating Curve= 0 ,0
Exp/Cntr=0.3,0.1

Type RM Length L Ch R = 1 ,85821.6 ,453.7,456.6,459.5
XS GIS Cut Line= 2
     1946042.315      244205.361     1946908.013      243032.872
#Sta/Elev= 30
       0 2854.69    89.8 2828.79   109.8 2825.72   129.8 2821.17   159.7 2823.83
   229.6 2833.18   249.6 2834.22   329.4 2823.53   349.4 2822.92   439.2 2811.98
   459.2 2810.82   499.1 2802.49     549 2789.64     559 2788.14     589  2787.3
     599  2787.3   918.4  2787.3   988.3 2789.16  1068.1 2794.09    1148 2805.16
    1168 2806.61  1257.8 2820.71  1277.8 2822.23  1307.7 2828.72  1347.6  2841.9
  1377.6 2849.84  1387.6 2849.83  1397.6 2851.96  1427.5 2860.38  1457.4 2867.33
#Mann= 3 , 0 , 0
       0      .1       0     599    .045       0   918.4      .1       0
Bank Sta=599,918.4
XS Rating Curve= 0 ,0
Exp/Cntr=0.3,0.1

Type RM Length L Ch R = 1 ,85364.6 ,442.5,437.9,434.3
XS GIS Cut Line= 2
     1946343.031      244430.139     1947275.555      243385.226
#Sta/Elev= 30
       0 2890.54      50 2886.67   180.1 2873.54   230.1 2858.79   250.1 2856.06
   280.1 2848.22   290.1 2844.63   360.1 2830.66   410.2 2818.76   460.2 2811.46
   540.2 2802.71   630.2 2788.32   640.2 2787.48   650.2  2787.3   960.4 2787.33
   970.4 2787.65   990.4 2791.25  1010.4 2796.19  1020.4 2799.62  1050.4 2806.86
  1130.4 2833.26  1140.4 2837.34  1150.4 2842.57  1160.4 2845.55  1170.4 2847.27
  1210.4 2862.06  1240.5 2870.82  1270.5 2875.39  1280.5 2875.92  1400.5 2876.88
#Mann= 3 , 0 , 0
       0      .1       0   640.2    .045       0   960.4      .1       0
Bank Sta=640.2,960.4
XS Rating Curve= 0 ,0
Exp/Cntr=0.3,0.1

Type RM Length L Ch R = 1 ,84926   ,728.2,718.3,707.5
XS GIS Cut Line= 3
     1946336.956      245301.912     1946895.863      244645.804
     1947551.971       243455.09
#Sta/Elev= 30
       0 2882.84    69.4 2857.92    89.2 2855.08   138.7 2842.58   188.2 2833.13
     208 2832.08   297.2 2817.56   336.8 2816.18   435.9 2829.82   455.7 2827.07
   554.8 2831.23   574.6 2828.65   683.6 2845.05   703.4 2841.97   802.4 2837.81
   822.3 2832.25   861.9  2831.3   911.9 2835.18   961.8 2834.61  1051.8 2818.73
  1131.8 2799.93  1281.7  2787.3  1691.6 2787.28  1701.6 2787.96  1761.6 2806.02
  1781.6    2810  1871.5 2854.96  1921.5 2866.55  2081.4 2866.92  2221.4 2857.67
#Mann= 3 , 0 , 0
       0      .1       0  1281.7    .045       0  1701.6      .1       0
Bank Sta=1281.7,1701.6
XS Rating Curve= 0 ,0
Exp/Cntr=0.3,0.1

Type RM Length L Ch R = 1 ,84208.6 ,618.1,599.7,581.2
XS GIS Cut Line= 3
     1947217.842      245636.042     1947731.186      244970.821
     1947980.264       243479.39
#Sta/Elev= 30
       0 2881.27     100 2879.64     140 2880.22   360.1 2871.47   400.1 2865.94
   440.1  2857.2   500.2  2847.4   550.2 2845.76   640.2 2832.92   670.2 2831.26
   730.2 2825.37   830.3 2809.69   850.2 2807.94   929.8 2796.22  1009.4 2787.39
  1496.2 2786.84  1745.5  2786.6  1765.4 2786.48  1785.3 2787.44    1845 2809.09
  1864.9 2814.67  1964.4 2825.33  2024.1  2830.5  2073.8 2831.54  2103.6 2831.09
  2163.3 2827.42    2233 2826.01  2262.8 2828.26  2342.4 2839.37  2352.4 2839.67
#Mann= 3 , 0 , 0
       0      .1       0  1496.2    .045       0  1745.5      .1       0
Bank Sta=1496.2,1745.5
XS Rating Curve= 0 ,0
Exp/Cntr=0.3,0.1

Type RM Length L Ch R = 1 ,83606.9 ,980.6,1017.9,1055.3
XS GIS Cut Line= 4
     1947715.998      245623.891     1948553.899       244445.71
     1948114.637      243919.731     1948235.417      242841.507
#Sta/Elev= 30
       0 2860.41   209.4 2853.88   239.3 2856.16     339 2843.97   408.8 2841.76
   448.7 2833.56   488.6 2833.35   538.4 2841.27     698 2851.25   767.7 2845.25
   807.6 2845.58   897.4 2831.93   937.2 2829.51  1196.5 2831.52  1445.8 2817.54
  1535.1 2802.65  1584.8 2788.37  1614.6 2786.48  2021.8  2786.5  2051.6 2788.54
  2091.3  2806.1  2190.8    2833  2210.7 2835.96  2240.5 2850.23  2260.4 2854.84
  2608.8 2844.04  2977.1 2846.03  3116.5 2828.61  3186.1 2830.15    3216 2834.84
#Mann= 3 , 0 , 0
       0      .1       0  1614.6    .045       0  2021.8      .1       0
Bank Sta=1614.6,2021.8
XS Rating Curve= 0 ,0
Exp/Cntr=0.3,0.1

Type RM Length L Ch R = 1 ,82588.3 ,680.4,661.7,642.6
XS GIS Cut Line= 4
     1948311.355      245332.288     1948838.672      244362.752
     1949481.979      243889.099     1949729.885      242817.207
#Sta/Elev= 30
       0 2872.59   119.3 2874.21   198.9 2871.37   367.9 2857.42   447.4 2845.19
   497.1 2850.44     696 2857.43     875 2837.33   944.6 2825.55  1063.9  2817.1
  1113.6 2818.18  1193.5 2812.26  1243.5  2801.9  1283.4 2788.78  1303.4 2786.52
  1313.4  2786.5  1692.8  2786.5  1722.8  2788.9  1782.7 2803.61  1852.6 2813.42
  1962.5 2819.13  2122.6 2814.52  2252.6 2815.39  2352.6  2804.9  2402.6 2803.42
  2502.6 2810.51  2672.7 2811.47  2882.7 2817.18  2942.7 2816.51  3002.7 2811.97
#Mann= 3 , 0 , 0
       0      .1       0  1303.4    .045       0  1692.8      .1       0
Bank Sta=1303.4,1692.8
XS Rating Curve= 0 ,0
Exp/Cntr=0.3,0.1

Type RM Length L Ch R = 1 ,81926.4 ,878.4,890.3,902.2
XS GIS Cut Line= 5
     1949164.903      245797.031     1949445.933      245309.539
     1949535.483      244855.394     1949729.828      243775.761
     1949757.991      242649.187
#Sta/Elev= 30
       0 2840.32   177.7 2834.27   266.5 2832.09   345.5 2832.16   394.9 2829.63
   454.1 2831.11   562.7 2830.52   789.2 2820.47   986.2 2813.93  1025.6 2807.85
  1035.6    2804  1065.5 2787.49  1075.4 2786.44  1085.4  2786.5  1663.8  2786.5
  1703.7 2788.04  1743.6 2799.81  1753.6 2800.23  1813.4 2817.48  1883.2 2828.28
  1903.2 2829.66  2042.8 2825.56  2122.6 2815.57  2202.4  2811.2  2371.9 2813.36
  2471.6 2808.96  2561.4 2807.52  3010.2 2811.68  3199.6 2801.15  3249.5 2802.13
#Mann= 3 , 0 , 0
       0      .1       0  1085.4    .045       0  1663.8      .1       0
Bank Sta=1085.4,1663.8
XS Rating Curve= 0 ,0
Exp/Cntr=0.3,0.1

Type RM Length L Ch R = 1 ,81035.6 ,956.1,972.8,989.5
XS GIS Cut Line= 4
     1949869.612      246140.273     1950018.451      245368.738
     1950551.488      244723.483     1951241.703      243547.945
#Sta/Elev= 30
       0  2854.1   129.3 2854.45   407.8 2836.85   576.9 2830.92   656.5 2830.15
   706.2 2825.62     746 2817.34   795.7 2811.06   845.5 2808.26   875.4 2808.96
   925.2 2795.52   945.2 2787.73   975.1  2786.5  1313.8  2786.5  1333.8 2786.49
  1363.6 2789.79  1433.4 2810.43  1483.2  2831.5  1513.1 2836.32  1692.4 2834.91
    1762 2830.59  1841.6 2822.78  1951.1 2818.29  2030.7 2818.52  2259.5 2825.35
  2408.8 2823.07  2597.8 2814.01    2757 2810.84  2856.5 2811.53  2985.9 2816.92
#Mann= 3 , 0 , 0
       0      .1       0   975.1    .045       0  1313.8      .1       0
Bank Sta=975.1,1313.8
XS Rating Curve= 0 ,0
Exp/Cntr=0.3,0.1

Type RM Length L Ch R = 1 ,80062.6 ,390.4,372,353.6
XS GIS Cut Line= 4
     1949911.672      246017.988     1950305.481       245958.52
      1950562.36      245740.552     1951223.568      245164.375
#Sta/Elev= 30
       0 2855.53   199.1 2843.86   209.1 2841.35     229 2819.12   258.9 2794.04
   268.8 2788.68   288.8 2786.49   294.6  2786.5   309.6  2786.5   338.5 2787.73
   348.5 2791.93   368.4 2808.89   388.3 2830.65   398.3 2833.37   457.7 2827.31
   527.1 2817.32   596.4 2812.92   695.5 2811.52   735.2 2813.02   755.1 2811.48
     785 2813.44  1014.2  2813.8  1183.6  2811.9  1313.2    2824  1343.1 2828.36
    1373 2834.82  1392.9 2836.94  1502.6 2831.88  1582.3  2835.5  1612.2 2835.26
#Mann= 3 , 0 , 0
       0      .1       0   294.6    .045       0   309.6      .1       0
Bank Sta=294.6,309.6
XS Rating Curve= 0 ,0
Exp/Cntr=0.3,0.1

Type RM Length L Ch R = 1 ,79690.6 ,180.3,180.8,181.2
XS GIS Cut Line= 2
     1950162.587      246605.765     1950509.794      246106.249
#Sta/Elev= 30
       0 2860.47    59.8 2858.45   179.5 2853.02   209.4 2850.95   229.4 2849.04
   239.3 2848.36   289.2 2845.61   299.2  2844.7   309.2 2842.96   319.1 2835.53
   329.1 2822.32   339.1 2808.13     349 2795.56     359    2788     369 2786.57
     379  2786.5     399  2786.5     414  2786.5   448.8 2786.53   458.7  2787.5
   468.7 2793.55   478.7 2801.56   488.7 2804.85   498.6 2805.66   548.5 2808.42
   558.5 2808.84   568.4 2808.68   578.4 2807.33   598.4 2803.67   608.3 2802.19
#Mann= 3 , 0 , 0
       0      .1       0     399    .045       0     414      .1       0
Bank Sta=399,414
XS Rating Curve= 0 ,0
Exp/Cntr=0.3,0.1

Type RM Length L Ch R = 1 ,79509.8 ,106.8,105.6,104.3
XS GIS Cut Line= 2
     1950292.606      246719.908     1950659.745      246213.892
#Sta/Elev= 30
       0 2857.32    99.2 2854.18     129 2852.91   168.7 2850.65   198.5 2849.68
   238.2  2847.8     258 2846.62   287.8 2843.56   297.7 2843.22   337.4 2839.08
   347.3 2835.99   357.2 2827.65   377.1 2805.88     387 2796.15   396.9 2790.36
   406.9 2789.14   422.3 2788.57   437.3 2787.67   456.5 2786.66   466.4  2788.2
   486.2 2796.14   496.2 2799.24   506.1 2801.78     516 2804.94   525.9 2806.38
   535.9 2806.94   545.8 2807.15   605.3 2804.59   615.2  2802.8   625.2 2799.69
#Mann= 3 , 0 , 0
       0      .1       0   422.3    .045       0   437.3      .1       0
Bank Sta=422.3,437.3
XS Rating Curve= 0 ,0
Exp/Cntr=0.3,0.1

Type RM Length L Ch R = 1 ,79404.3 ,176.4,173.2,170
XS GIS Cut Line= 3
     1950397.025      246796.956     1950695.606      246333.067
      1950708.42      246316.408
#Sta/Elev= 30
       0 2853.86    49.3 2853.38   128.1 2854.16   157.6 2854.18   187.2 2853.79
   226.6 2852.43   246.3 2851.33   285.7 2848.48   305.4 2846.41   334.9 2841.01
   354.6 2837.76   364.5 2834.09   374.4 2832.15   384.2 2822.49     394 2809.26
   403.9 2797.78   413.8 2791.15   423.6 2789.48   431.9 2788.62   446.9 2787.42
   453.2    2787     463 2787.08   472.9 2789.15   482.7 2794.05   492.6 2796.04
   502.4 2799.47     532 2812.41   541.8 2814.16   551.7 2813.33   572.7 2810.45
#Mann= 3 , 0 , 0
       0      .1       0   431.9    .045       0   446.9      .1       0
Bank Sta=431.9,446.9
XS Rating Curve= 0 ,0
Exp/Cntr=0.3,0.1

Type RM Length L Ch R = 1 ,79231.1 ,155,144.8,134.5
XS GIS Cut Line= 2
     1950642.087      246826.412      1950840.88      246391.123
#Sta/Elev= 30
       0 2832.34    39.9 2827.64    59.8 2825.63    79.8 2824.01   119.6 2819.82
   139.6 2817.55   159.5 2814.42   169.5 2813.07   179.4 2812.39   189.4 2811.24
   229.3 2805.08   239.3 2803.25   249.2  2801.9   269.2  2798.4   279.1 2797.22
   299.1 2793.78     319 2789.62   336.6 2785.17     339 2784.55   348.9 2783.67
   351.6 2784.34   358.9 2786.14   368.9    2791   378.8 2791.75   388.8 2794.16
   418.7 2803.11   428.7  2805.3   438.7 2804.87   458.6 2800.57   478.5 2796.51
#Mann= 3 , 0 , 0
       0      .1       0   336.6    .045       0   351.6      .1       0
Bank Sta=336.6,351.6
XS Rating Curve= 0 ,0
Exp/Cntr=0.3,0.1

Type RM Length L Ch R = 1 ,79086.3 ,258.9,275.1,291.4
XS GIS Cut Line= 3
     1950819.714      246857.962     1950924.205      246759.981
     1950924.653      246424.212
#Sta/Elev= 30
       0 2807.77    28.6 2805.33    57.3 2804.74    66.8 2803.89   124.1 2792.98
   153.1 2789.11     163 2788.22   172.9  2787.9   202.5 2787.89   232.1 2787.07
     242 2785.79   261.8 2781.56   301.2  2770.6     321  2765.6   330.9 2765.07
   340.8 2763.23   350.6  2762.2   352.5  2762.5   360.5 2763.75   367.5 2766.95
   370.4 2768.27   380.3 2773.92   390.1 2778.67     400 2782.37   409.9 2785.26
   439.5 2788.46   449.4    2789   459.3 2788.98   469.1 2788.23     479 2786.48
#Mann= 3 , 0 , 0
       0      .1       0   352.5    .045       0   367.5      .1       0
Bank Sta=352.5,367.5
XS Rating Curve= 0 ,0
Exp/Cntr=0.3,0.1

Type RM Length L Ch R = 1 ,78811.1 ,341,330.9,324.3
XS GIS Cut Line= 2
     1950885.119      246988.421     1951546.938      246211.181
#Sta/Elev= 30
       0 2830.75      20 2831.96      30  2830.1      50 2823.53      60 2822.74
    70.1 2820.04    90.1 2812.85   140.1  2791.4   170.1 2783.43   210.2  2781.1
   270.2 2782.23   300.2 2773.04   330.3 2752.67   350.3 2737.18   360.3 2734.19
   419.3 2733.97   434.3 2733.04   460.4 2732.28   470.4 2732.64   530.4 2741.45
   580.5 2745.15   680.6 2746.04   720.6 2750.02   770.6 2761.59   840.7 2772.79
   860.7 2777.59   940.8 2791.54   960.8 2796.22   990.8 2806.53  1020.8 2813.94
#Mann= 3 , 0 , 0
       0      .1       0   419.3    .045       0   434.3      .1       0
Bank Sta=419.3,434.3
XS Rating Curve= 0 ,0
Exp/Cntr=0.3,0.1

Type RM Length L Ch R = 1 ,78480.3 ,407.5,406.9,402.8
XS GIS Cut Line= 3
     1951300.222      247262.944     1951401.032      246867.463
     1951567.091      246484.645
#Sta/Elev= 30
       0 2829.92    19.9 2823.81    29.9 2822.68    39.8 2820.51    99.5  2803.1
   119.4 2796.06   129.4 2793.35   139.4  2792.1   199.1 2769.81     219 2761.62
     229 2760.38   258.8 2748.11   308.6 2730.61   338.4  2725.8   388.2 2720.36
   398.2 2719.92   400.6 2720.15   415.6 2722.06     428 2722.82   457.8 2728.48
   507.5  2735.8   547.2 2738.08   626.7 2741.12   656.5 2744.26   676.4 2747.57
   686.3 2750.53   706.2  2759.9   765.8 2772.94   775.7 2774.28   825.4 2775.01
#Mann= 3 , 0 , 0
       0      .1       0   400.6    .045       0   415.6      .1       0
Bank Sta=400.6,415.6
XS Rating Curve= 0 ,0
Exp/Cntr=0.3,0.1

Type RM Length L Ch R = 1 ,78073.3 ,378,392.9,407.9
XS GIS Cut Line= 3
     1951640.881      247394.358     1951711.184      247301.692
     1951872.277      246608.377
#Sta/Elev= 30
       0 2809.43    38.8 2802.92    67.8 2794.06    96.9 2789.49   126.2 2781.92
   175.6 2767.55   195.4 2764.31   264.6 2742.08   274.5  2739.5   284.4  2738.4
   323.9 2723.99   343.7 2717.93   373.4 2712.37   383.2 2712.08     403 2707.95
   409.9 2707.59   412.9 2707.44   424.9 2709.66   462.3 2718.59   482.1 2720.45
   541.4 2734.72   561.2 2737.26     581 2737.43   590.8 2739.55     660 2764.55
   669.9  2765.4   679.8  2768.1     749 2789.32   768.8 2792.11   828.1 2807.44
#Mann= 3 , 0 , 0
       0      .1       0   409.9    .045       0   424.9      .1       0
Bank Sta=409.9,424.9
XS Rating Curve= 0 ,0
Exp/Cntr=0.3,0.1

Type RM Length L Ch R = 1 ,77680.3 ,375.7,371.8,367.9
XS GIS Cut Line= 3
     1951766.301      247489.711     1952084.234      247231.624
     1952402.167      246973.537
#Sta/Elev= 30
       0 2831.25      10  2828.2      40 2821.03    89.9 2804.62    99.9  2802.2
   119.8 2794.93   139.8 2789.39   169.8 2779.65   199.8 2768.94   219.7 2759.49
   249.7 2747.51   269.7 2743.25   299.6 2731.53   319.6 2721.85   339.6 2716.47
     402 2703.58     417 2700.23   419.5 2699.58   429.5    2700   529.4 2712.48
   559.3 2714.21   609.3 2718.92   619.2 2720.68   649.2 2730.68   679.2 2742.29
   699.2 2746.08   729.1 2759.29   749.1 2766.25     779 2778.36     819 2788.01
#Mann= 3 , 0 , 0
       0      .1       0     402    .045       0     417      .1       0
Bank Sta=402,417
XS Rating Curve= 0 ,0
Exp/Cntr=0.3,0.1

Type RM Length L Ch R = 1 ,77308.5 ,433.9,449.6,465.3
XS GIS Cut Line= 2
     1952089.146      247773.588     1952641.226      247139.335
#Sta/Elev= 30
       0 2785.89    29.7 2783.02    49.5 2777.58    69.2 2769.58    79.1 2768.16
      89 2764.23   128.6 2740.52   138.5 2732.28   148.4 2725.77   168.2 2715.83
   178.1 2712.66   296.8  2700.3   428.5 2691.01   435.3 2690.75   443.5 2691.52
     465 2695.78   474.8 2698.76   494.6 2705.43   514.4 2714.19   573.8 2735.72
   593.6 2740.14   613.3 2747.24   633.1 2756.41   682.6 2771.23   702.4 2776.17
     732 2781.03   751.8 2787.05   771.6 2791.42   811.2 2798.23   840.9 2801.16
#Mann= 3 , 0 , 0
       0      .1       0   428.5    .045       0   443.5      .1       0
Bank Sta=428.5,443.5
XS Rating Curve= 0 ,0
Exp/Cntr=0.3,0.1

Type RM Length L Ch R = 1 ,76858.7 ,354.4,361.4,368.5
XS GIS Cut Line= 2
     1952148.144      247863.365     1953022.561      247722.148
#Sta/Elev= 30
       0 2775.77    19.9 2769.72    39.8  2759.3    99.5  2738.3   109.5  2734.2
   119.4 2729.02   159.2  2716.6   189.1 2710.27     199 2706.85     209 2704.85
   268.7 2694.16   278.7 2691.37   298.6 2689.44   358.3 2685.91   483.1 2682.01
   497.6 2681.71   498.1 2681.75   507.6 2682.43   527.5 2691.53   587.2 2709.53
   607.1 2718.04   636.9 2725.61   686.7 2736.02   696.6 2739.12   756.4 2752.54
   766.3 2755.24   776.3 2760.12   845.9 2777.61   855.9 2782.41   885.8 2789.67
#Mann= 3 , 0 , 0
       0      .1       0   483.1    .045       0   498.1      .1       0
Bank Sta=483.1,498.1
XS Rating Curve= 0 ,0
Exp/Cntr=0.3,0.1

Type RM Length L Ch R = 1 ,76497.3 ,431.7,416.9,402
XS GIS Cut Line= 2
     1952116.982      248059.831     1952973.314      248160.953
#Sta/Elev= 30
       0 2825.76    49.6 2797.01    59.5 2790.91    69.4 2784.07   128.8 2765.91
   138.8 2762.42   148.7 2756.85     218 2735.78     228  2729.7   297.3 2708.52
   307.2 2702.95   317.2 2699.67   376.6 2682.44   386.5 2680.76   392.9 2680.53
   396.4  2680.4   407.9  2680.4   436.1  2680.9   515.4 2688.49   535.2 2690.76
   574.8 2698.81   624.4  2712.5   634.3  2715.8   644.2 2720.07   703.7 2737.54
   713.6 2741.16   723.5 2746.65   792.9 2767.09   802.8 2772.07   862.3 2786.05
#Mann= 3 , 0 , 0
       0      .1       0   392.9    .045       0   407.9      .1       0
Bank Sta=392.9,407.9
XS Rating Curve= 0 ,0
Exp/Cntr=0.3,0.1

Type RM Length L Ch R = 1 ,76080.3 ,394.6,400,405.4
XS GIS Cut Line= 3
     1952302.085      248682.929     1952654.375      248474.165
     1953006.664      248265.401
#Sta/Elev= 30
       0  2747.3      30 2738.46      40 2734.65    49.9 2729.91    59.9 2727.11
   129.8  2711.4   139.8  2707.3   219.7 2688.32   239.7 2682.73   249.7 2680.71
   259.7  2680.4   289.6  2680.4     402  2680.4   449.4 2680.49   459.4  2681.2
   489.4 2686.23   509.4 2691.46   529.4 2700.33   549.3 2707.33   599.3 2727.09
   619.2 2736.61   629.2  2739.2   649.2 2746.79   669.2 2755.18   699.2 2764.16
   709.1  2769.3   729.1 2774.88     789 2788.62     809 2795.84     819 2797.92
#Mann= 3 , 0 , 0
       0      .1       0   289.6    .045       0     402      .1       0
Bank Sta=289.6,402
XS Rating Curve= 0 ,0
Exp/Cntr=0.3,0.1

Type RM Length L Ch R = 1 ,75680.3 ,349.5,346.1,342.6
XS GIS Cut Line= 3
     1952407.699      248963.952     1952799.704      248845.534
     1953191.708      248727.116
#Sta/Elev= 30
       0 2767.08      10 2763.29      20 2758.54      30 2752.93    99.9 2727.59
   109.9 2720.75   149.8 2707.54   179.8 2696.54   199.8 2686.01   209.7 2682.63
   219.7 2680.75   229.7  2680.4   239.7  2680.4   499.4  2680.4   509.4 2680.43
   519.4  2681.6   529.4 2686.69   599.3 2705.15   609.3 2709.93   619.2 2713.92
   649.2 2724.93   679.2 2737.13   689.2  2742.4   699.2 2748.53   729.1 2758.65
   749.1 2763.33   769.1 2766.65     779 2769.02     799 2770.35     819 2770.05
#Mann= 3 , 0 , 0
       0      .1       0   239.7    .045       0   499.4      .1       0
Bank Sta=239.7,499.4
XS Rating Curve= 0 ,0
Exp/Cntr=0.3,0.1

Type RM Length L Ch R = 1 ,75334.2 ,417.5,417.8,417.9
XS GIS Cut Line= 3
     1952538.417      249348.709     1952908.931      249174.479
     1953278.042      248996.285
#Sta/Elev= 30
       0 2760.99      20 2764.15    39.9 2766.55    49.9 2767.48    59.9 2767.16
    99.9 2762.53   109.8 2761.03   129.8 2756.75   139.8  2753.5   149.8 2747.22
   159.8 2743.51   179.8 2734.98   189.7 2729.49   199.7 2722.94   219.7  2707.2
   229.7 2697.77   239.7    2686   249.6  2681.1   259.6  2680.3   269.6  2680.4
   569.4  2680.4   579.4 2680.45   589.4 2681.06   609.4 2685.16   659.4 2693.15
   669.4 2694.22   729.3 2699.67   739.3 2700.15   759.3 2699.89   819.3  2704.2
#Mann= 3 , 0 , 0
       0      .1       0   269.6    .045       0   569.4      .1       0
Bank Sta=269.6,569.4
XS Rating Curve= 0 ,0
Exp/Cntr=0.3,0.1

Type RM Length L Ch R = 1 ,74916.1 ,1200.7,1218.8,1231.4
XS GIS Cut Line= 4
     1952118.403      249742.377     1952842.856       249639.86
     1953768.045      249185.161     1954547.674      248639.371
#Sta/Elev= 30
       0 2805.51     178 2807.71   227.4 2805.24   296.6 2796.32   306.5 2793.93
   326.3 2782.15   385.6 2758.59   405.4 2747.12   484.5 2717.63   563.6 2705.57
   642.7 2696.76   791.7 2682.03   831.8  2680.4   841.8  2680.4  1332.2  2680.4
  1372.2 2681.64  1452.3 2715.36  1522.4 2736.46  1552.4  2749.7  1622.4 2771.05
  1642.4 2775.02  1891.4 2794.25  1960.8 2802.84  2149.2 2816.17  2218.6 2811.54
  2297.9 2802.24  2416.8 2797.56  2545.7 2775.16    2625 2764.52  2714.2 2745.66
#Mann= 3 , 0 , 0
       0      .1       0   841.8    .045       0  1332.2      .1       0
Bank Sta=841.8,1332.2
XS Rating Curve= 0 ,0
Exp/Cntr=0.3,0.1

Type RM Length L Ch R = 1 ,73696.5 ,526.5,517,507.4
XS GIS Cut Line= 3
     1952360.647      250124.727     1953612.112      250243.191
     1955307.058      249508.107
#Sta/Elev= 30
       0 2778.08   139.7  2770.5   259.4 2748.42   309.3 2735.36     449 2683.45
   488.9  2675.5   508.8  2675.5   927.8  2675.5   957.8 2675.74  1127.4 2718.71
  1237.1  2754.3    1277 2759.06  1466.8 2740.28  1516.7 2739.56  1576.6 2730.47
  1706.4  2728.8  1836.3 2732.14  1866.2 2737.68    2016 2742.68  2125.9 2753.53
  2285.7 2759.99  2315.6 2764.82  2465.4 2762.21  2565.3 2764.66    2795  2751.2
  2814.9 2747.03  2924.8 2704.62  2984.7 2696.62  3004.7 2697.22  3104.5 2734.56
#Mann= 3 , 0 , 0
       0      .1       0   508.8    .045       0   927.8      .1       0
Bank Sta=508.8,927.8
XS Rating Curve= 0 ,0
Exp/Cntr=0.3,0.1

Type RM Length L Ch R = 1 ,73179.3 ,449.5,449.2,449
XS GIS Cut Line= 3
     1952167.069      251026.593      1953446.48       250590.75
     1954138.908      250488.819
#Sta/Elev= 30
       0 2806.99    59.6 2794.93   119.3 2785.46     169  2782.2   228.6 2775.18
   407.5 2762.61   606.2 2756.28   695.7 2749.67   715.6 2744.78   735.4 2742.35
   785.1 2740.36   874.6 2688.54   884.5 2679.81   894.4 2676.89   914.3  2675.5
  1212.5  2675.5  1252.2 2676.49  1301.9 2688.02  1381.6 2711.76  1401.6 2720.19
  1471.6 2740.56  1481.6 2745.47  1551.6  2763.7  1561.6 2768.62  1591.6 2776.27
  1631.6 2782.15  1701.6 2796.26  1721.6 2798.12  1981.5  2800.6  2051.5 2803.26
#Mann= 3 , 0 , 0
       0      .1       0   914.3    .045       0  1212.5      .1       0
Bank Sta=914.3,1212.5
XS Rating Curve= 0 ,0
Exp/Cntr=0.3,0.1

Type RM Length L Ch R = 1 ,72729.7 ,244.3,255.5,266.7
XS GIS Cut Line= 2
     1952469.347      251399.169      1954103.76      250826.246
#Sta/Elev= 30
       0 2761.19    39.8 2761.51    99.5 2766.23   139.4 2771.68   238.9  2766.5
   378.2 2743.44   398.1 2737.71     438 2730.25   487.7 2718.68   577.3 2704.44
   716.7 2684.83   736.6 2681.48   746.5 2678.33   776.4  2675.5  1055.1  2675.5
    1075  2675.5  1094.9 2679.52  1154.6 2701.62  1174.5    2712  1214.3 2724.91
  1244.2 2732.48  1254.2 2737.06  1323.8 2758.43  1343.7 2767.57  1373.6 2777.39
  1393.5 2785.82  1403.4 2788.16  1443.3 2792.23  1473.1 2792.68  1731.9 2787.78
#Mann= 3 , 0 , 0
       0      .1       0   776.4    .045       0  1055.1      .1       0
Bank Sta=776.4,1055.1
XS Rating Curve= 0 ,0
Exp/Cntr=0.3,0.1

Type RM Length L Ch R = 1 ,72473.6 ,775.9,767.2,758.6
XS GIS Cut Line= 4
     1952525.585      251529.219     1953069.573      251309.358
     1953717.124      251413.229     1954230.295      251536.249
#Sta/Elev= 30
       0 2786.74   119.3 2791.13   218.8 2792.52   238.7 2790.57   258.6  2782.8
   328.2 2761.63   348.1 2753.05   387.8 2741.93   437.6 2729.77   517.1 2716.23
   566.8 2705.12   596.7 2693.96   616.6 2681.59   636.4 2676.17   646.4  2675.5
   994.2  2675.5    1014 2675.49  1033.9 2676.91  1153.1 2692.62    1183 2698.92
  1252.5 2710.28  1272.4  2715.6  1342.1 2729.76  1352.1 2734.08    1362 2736.54
  1451.7  2755.5  1541.3 2769.86    1611 2779.41  1620.9 2782.12  1770.3 2800.61
#Mann= 3 , 0 , 0
       0      .1       0   646.4    .045       0   994.2      .1       0
Bank Sta=646.4,994.2
XS Rating Curve= 0 ,0
Exp/Cntr=0.3,0.1

Type RM Length L Ch R = 1 ,71706.4 ,779.6,796.9,814.2
XS GIS Cut Line= 2
     1952465.833       252288.43     1954550.147      251852.587
#Sta/Elev= 30
       0 2807.21      60  2805.7     140 2808.65   239.9  2835.3   279.9 2840.51
   319.9 2841.55   369.9 2836.76   379.9 2834.89   439.9 2807.42   549.8 2768.28
   559.8  2762.2   659.8 2735.02   719.8  2731.8   759.8 2707.66   859.8 2679.12
   889.8  2675.5  1199.7  2675.5  1229.6 2675.78  1259.6  2682.2  1369.6 2720.02
  1389.6 2729.88  1479.6 2762.89  1499.6  2773.2  1579.6 2782.77  1649.5 2784.79
  1769.5  2800.5  1829.5 2815.29  1899.5 2827.93  2079.4 2876.05  2129.4 2886.06
#Mann= 3 , 0 , 0
       0      .1       0   889.8    .045       0  1199.7      .1       0
Bank Sta=889.8,1199.7
XS Rating Curve= 0 ,0
Exp/Cntr=0.3,0.1

Type RM Length L Ch R = 1 ,70908.9 ,811.8,828.3,844.7
XS GIS Cut Line= 2
     1952743.507      252436.054     1954286.532      253402.642
#Sta/Elev= 30
       0 2793.06   140.1 2797.43   190.1 2797.31   210.1 2792.05   230.1 2781.99
   260.1 2770.94   280.1 2766.27   320.1 2751.71   340.1 2746.35   420.2 2726.26
   500.2  2714.2   540.2 2706.25   600.3 2688.84   620.3 2680.95   650.3 2675.75
   809.7  2675.4   960.4  2675.5   980.4 2675.49  1000.4  2678.6  1070.5 2702.45
  1140.5 2735.04  1170.5 2746.08  1180.5  2752.9  1200.5 2759.92  1290.6 2784.83
  1380.6 2801.68  1410.6 2805.27  1500.6 2809.62  1710.7 2813.22  1820.8 2816.51
#Mann= 3 , 0 , 0
       0      .1       0   650.3    .045       0   960.4      .1       0
Bank Sta=650.3,960.4
XS Rating Curve= 0 ,0
Exp/Cntr=0.3,0.1

Type RM Length L Ch R = 1 ,70080.3 ,1181.9,1156.2,1130.7
XS GIS Cut Line= 3
     1952486.922      252446.599     1952720.167      253248.632
     1952855.983       253704.92
#Sta/Elev= 30
       0 2802.92   248.6  2797.8   278.4 2795.89   288.4 2794.24   328.1 2781.55
     348 2778.86   427.6 2759.58   437.5 2758.89   517.1 2734.02     527 2732.84
     537 2730.06   546.9 2725.67   556.8 2720.18   596.6  2694.1   616.5 2683.89
   626.4 2680.27   636.4 2679.33   646.3 2676.12   656.3  2675.5   964.2  2675.5
     984 2675.86  1023.7 2682.48    1103 2704.24    1113 2704.91  1202.2  2727.8
  1222.1 2730.68  1241.9 2734.97  1251.8 2734.96  1301.4 2725.53  1311.3 2726.04
#Mann= 3 , 0 , 0
       0      .1       0   656.3    .045       0   964.2      .1       0
Bank Sta=656.3,964.2
XS Rating Curve= 0 ,0
Exp/Cntr=0.3,0.1

Type RM Length L Ch R = 1 ,68923   ,2120.5,2109.6,2097.6
XS GIS Cut Line= 4
     1951063.402      253687.346     1952318.208      253884.178
      1952652.12      253701.405     1954605.691      253947.077
#Sta/Elev= 30
       0 2782.13     170 2777.97     310 2767.38     440 2734.04   510.1 2706.61
   570.1  2688.6   590.1 2679.55   630.1  2675.5  1030.1  2675.5  1040.1 2675.49
  1070.1 2676.84  1120.1 2684.01  1190.1 2701.82  1240.2 2709.84    1319 2710.69
  1514.2 2704.44  1670.8 2704.65  1710.8 2710.82  1840.7  2719.1  2030.6 2745.89
  2170.5 2751.33  2350.4 2776.42  2510.4 2786.07  2650.3 2785.54  2860.2  2802.1
  2970.1 2804.03    3140 2813.46  3299.9 2813.53  3389.9 2808.68  3619.8 2766.03
#Mann= 3 , 0 , 0
       0      .1       0   630.1    .045       0  1030.1      .1       0
Bank Sta=630.1,1030.1
XS Rating Curve= 0 ,0
Exp/Cntr=0.3,0.1

Type RM Length L Ch R = 1 ,66812.1 ,412.3,408.5,404.7
XS GIS Cut Line= 4
     1951010.679      255437.749     1952338.492      255408.007
     1953170.489      254991.111     1954623.959      254819.132
#Sta/Elev= 30
       0 2808.71   109.8 2823.04   159.8  2810.2   379.5 2772.56   459.4 2783.13
     689 2776.72   788.9  2759.4   958.7 2711.09  1088.5 2728.61  1228.3 2738.65
  1328.2 2725.22  1478.2 2682.12  1518.3 2675.54  1528.3  2675.5  1958.6  2675.5
  1998.6 2676.29  2088.6 2687.39  2178.7 2704.27  2238.7 2720.32  2298.6 2729.35
  2527.6 2752.08  2637.1 2741.04  2796.4 2773.13    2886 2777.34    3115 2797.39
  3234.5 2797.74  3393.8  2782.9  3503.3 2777.88    3563  2779.5  3722.4  2794.7
#Mann= 3 , 0 , 0
       0      .1       0  1518.3    .045       0  1958.6      .1       0
Bank Sta=1518.3,1958.6
XS Rating Curve= 0 ,0
Exp/Cntr=0.3,0.1

Type RM Length L Ch R = 1 ,66403.4 ,371.6,374,374.8
XS GIS Cut Line= 3
     1952539.845       255836.76     1953012.982      255494.589
     1953541.034      255118.428
#Sta/Elev= 30
       0 2781.06    29.7 2780.08    49.5 2778.17    89.1 2767.26   118.8 2755.34
   138.6 2750.34   197.9 2727.64   217.7 2718.26   247.4 2708.18   296.9 2695.29
   316.7 2687.67   346.4 2678.57   356.3  2676.3   366.2 2675.57   376.1  2675.5
   713.6 2675.96   743.5 2679.87   753.5 2683.88   773.4 2694.58   803.3 2703.38
   893.1 2719.87     923 2728.57     943 2731.64   982.9 2741.52  1002.8 2748.85
  1052.7  2761.5  1152.4 2774.18  1182.4 2779.52  1202.3 2784.72  1232.2 2789.38
#Mann= 3 , 0 , 0
       0      .1       0   366.2    .045       0   713.6      .1       0
Bank Sta=366.2,713.6
XS Rating Curve= 0 ,0
Exp/Cntr=0.3,0.1

Type RM Length L Ch R = 1 ,66028.8 ,124.6,125,126.9
XS GIS Cut Line= 6
     1952666.544      256140.421     1952987.908      255941.858
     1953147.559      255850.325     1953218.361      255811.432
     1953292.055      255785.067     1953903.366      255439.316
#Sta/Elev= 30
       0 2792.08   159.1 2787.61   188.9 2783.82   208.8 2776.23   248.5 2747.05
   278.4 2734.48     328 2708.49     338 2700.45   347.9 2695.12   357.9 2691.71
   397.6 2679.34   417.5 2677.35   504.2 2677.97   519.2 2677.71   534.5 2678.84
   552.8 2676.76   627.5 2678.84   642.7 2676.15   681.8 2679.77   740.8 2681.15
   780.3 2686.16   790.2 2690.57   859.5 2711.12     899 2729.45  1057.3 2785.16
  1077.1 2794.94  1106.8 2803.29  1146.3 2807.61  1225.5 2811.53  1423.3  2807.5
#Mann= 3 , 0 , 0
       0      .1       0   504.2    .045       0   519.2      .1       0
Bank Sta=504.2,519.2
XS Rating Curve= 0 ,0
Exp/Cntr=0.3,0.1

Type RM Length L Ch R = 1 ,65903.7 ,208.1,208.5,208.8
XS GIS Cut Line= 2
      1952788.71      256190.825     1953643.017      255729.499
#Sta/Elev= 30
       0 2789.14    59.4 2786.33    89.2 2778.75   128.8 2762.73   168.4 2740.03
   178.3 2733.58   188.2 2724.49     218 2710.01   227.9 2706.87   237.8 2706.24
   257.6 2708.96   267.5 2706.28   277.4 2691.76   287.3 2682.72   297.2 2675.93
   346.8  2652.2   366.6 2650.39   414.6  2650.4   429.6  2650.4   495.4 2651.58
   624.2 2670.02   673.7 2685.87   713.3 2696.24   733.1 2704.51   812.4 2728.72
   832.2 2737.32   881.7 2753.86   911.5 2761.34   931.3 2770.63   970.9 2784.45
#Mann= 3 , 0 , 0
       0      .1       0   414.6    .045       0   429.6      .1       0
Bank Sta=414.6,429.6
XS Rating Curve= 0 ,0
Exp/Cntr=0.3,0.1

Type RM Length L Ch R = 1 ,65695.2 ,383.3,407.7,432.1
XS GIS Cut Line= 4
     1952834.953      256244.982     1953095.406       256251.48
     1953607.066      255983.948     1953930.064      256057.553
#Sta/Elev= 30
       0 2788.61      29 2788.38    67.6 2775.51   115.8 2753.75   144.7 2743.09
   173.7 2719.86     193  2708.3   202.6 2705.78   241.2  2706.5   260.5 2704.35
   270.5 2700.37   280.4 2692.06   290.4 2687.39   350.1 2664.74     380 2658.13
   459.6 2647.95   469.6  2647.9   478.6  2648.1   493.6 2648.47   539.3  2652.1
     589 2658.61   738.4 2680.86   788.1 2693.25     818 2706.34   837.9 2721.51
   857.4  2725.2  1003.6 2743.05  1071.8 2746.26  1130.2 2754.08  1169.2 2755.02
#Mann= 3 , 0 , 0
       0      .1       0   478.6    .045       0   493.6      .1       0
Bank Sta=478.6,493.6
XS Rating Curve= 0 ,0
Exp/Cntr=0.3,0.1

Type RM Length L Ch R = 1 ,65287.5 ,407,407.2,407.3
XS GIS Cut Line= 3
     1952748.557      256251.267     1953085.581       256411.45
      1953701.11      256797.383
#Sta/Elev= 30
       0 2793.24   117.8 2788.26   127.7 2785.59   137.5  2777.2   176.8 2757.05
     216 2732.88   225.9 2722.88   255.3 2707.89   265.1 2706.04   353.5 2704.36
   393.1 2689.97   422.9 2674.86   472.7 2654.28   502.5 2643.88   513.8 2641.83
   522.4 2641.45   528.8 2642.38   552.3 2647.45     622 2657.99   681.7 2673.08
   701.6 2680.96   721.5 2686.53   781.2 2695.97   870.8 2720.54   890.7 2727.87
   940.4 2738.65   970.3    2747  1059.9 2779.18  1079.8 2788.33  1099.7 2792.17
#Mann= 3 , 0 , 0
       0      .1       0   513.8    .045       0   528.8      .1       0
Bank Sta=513.8,528.8
XS Rating Curve= 0 ,0
Exp/Cntr=0.3,0.1

Type RM Length L Ch R = 1 ,64880.3 ,389.2,378.6,368.1
XS GIS Cut Line= 3
     1952641.764      256610.119     1952987.159      256830.102
     1953332.553      257050.086
#Sta/Elev= 30
       0 2769.68      20 2762.31      40 2752.64    69.9 2733.39    89.9  2714.7
   109.9 2702.44   119.8 2697.21   129.8 2694.22   139.8 2693.59   189.8 2693.05
   199.8 2690.76   279.7 2663.02   329.6 2651.98   359.6 2649.45   389.5 2642.43
     402 2640.53   409.5 2640.09     417 2640.32   459.4  2643.9   499.4 2652.66
   519.4  2655.6   559.3 2662.91   569.3 2665.61   629.2 2677.12   649.2 2681.91
   669.2  2689.5   699.2 2696.31   729.1 2702.18   749.1  2704.5     819 2703.68
#Mann= 3 , 0 , 0
       0      .1       0     402    .045       0     417      .1       0
Bank Sta=402,417
XS Rating Curve= 0 ,0
Exp/Cntr=0.3,0.1

Type RM Length L Ch R = 1 ,64501.5 ,417.3,419.8,422.3
XS GIS Cut Line= 2
     1952410.522      257121.842     1953332.049      257214.285
#Sta/Elev= 30
       0 2783.85    49.8 2775.01    69.7 2769.52   129.5 2757.62   149.4 2751.11
   179.3 2743.69   199.2 2737.56   209.1 2733.69     229 2720.38   268.9 2703.08
   288.8 2693.61   308.7 2678.66   358.5 2653.09   388.4 2639.93   396.1 2639.63
   398.3 2639.54   411.1 2640.13   497.9 2647.81   597.5 2652.74   627.4 2655.07
   677.2 2663.69   707.1 2670.63     717 2675.86   786.7 2694.96   796.7 2699.59
   826.6 2706.27   846.5 2707.04   906.2 2705.56   916.2  2706.7   926.2  2710.1
#Mann= 3 , 0 , 0
       0      .1       0   396.1    .045       0   411.1      .1       0
Bank Sta=396.1,411.1
XS Rating Curve= 0 ,0
Exp/Cntr=0.3,0.1

Type RM Length L Ch R = 1 ,64081.6 ,381.4,400.9,421.2
XS GIS Cut Line= 3
      1952455.53      257463.743     1952544.378      257496.206
     1953388.433      257675.611
#Sta/Elev= 30
       0 2753.08    47.3 2745.36    94.6 2732.29   134.3 2714.52   173.9 2693.96
   183.9 2687.75     283 2655.59   312.8 2652.22   362.4 2651.02   372.3 2649.19
   392.2 2641.92   406.9 2639.61     412 2639.47   421.9 2640.21   441.7 2643.49
   481.4 2647.22   501.2 2650.78     531 2658.91   590.5 2671.03   610.4  2677.1
   669.9 2689.62   689.7 2695.31   759.1 2693.96     769 2698.87   788.9 2705.74
   838.5 2725.47   848.4 2732.33   858.3 2737.27     898 2753.27   957.5    2773
#Mann= 3 , 0 , 0
       0      .1       0   406.9    .045       0   421.9      .1       0
Bank Sta=406.9,421.9
XS Rating Curve= 0 ,0
Exp/Cntr=0.3,0.1
